--- Stebenka.prj (project) ---

Proj Title=Stebenka
Current Plan=p08
Default Exp/Contr=0.3,0.1
SI Units
Geom File=g04
Flow File=f01
Unsteady File=u01
Unsteady File=u02
Unsteady File=u03
Unsteady File=u04
Unsteady File=u05
Plan File=p01
Plan File=p06
Plan File=p07
Plan File=p08
Y Axis Title=Elevation
X Axis Title(PF)=Main Channel Distance
X Axis Title(XS)=Station
BEGIN DESCRIPTION:
END DESCRIPTION:
DSS File=dss
DSS Export Rating Curves= 0
DSS Export Rating Curve Sorted= 0
DSS Export Volume Flow Curves= 0
DXF OffsetX= 0
DXF OffsetY= 0
DXF ScaleX= 1
DXF ScaleY= 10

--- Stebenka.p08 (plan) ---

Plan Title=ust_Q5
Program Version=5.07
Short Identifier=ust_Q5
Simulation Date=01SEP2008,0000,01SEP2008,0200
Geom File=g04
Flow File=u05
Subcritical Flow
K Sum by GR= 0
Std Step Tol= 0.003
Critical Tol= 0.003
Num of Std Step Trials= 20
Max Error Tol= 0.1
Flow Tol Ratio= 0.001
Split Flow NTrial= 30
Split Flow Tol= 0.006
Split Flow Ratio= 0.02
Log Output Level= 0
Friction Slope Method= 1
Unsteady Friction Slope Method= 2
Unsteady Bridges Friction Slope Method= 1
Parabolic Critical Depth
Global Vel Dist= 0 , 0 , 0
Global Log Level= 0
CheckData=True
Encroach Param=-1 ,0,0, 0
Computation Interval=1SEC
Output Interval=15MIN
Instantaneous Interval=15MIN
Mapping Interval=15MIN
Computation Time Step Use Courant=        0
Computation Time Step Use Time Series=    0
Computation Time Step Count To Double=0
Computation Time Step Max Doubling=0
Computation Time Step Max Halving=0
Computation Time Step Residence Courant=0
Run HTab=-1
Run UNet=-1
Run Sediment= 0
Run PostProcess=-1
Run WQNet= 0
Run RASMapper= 0
UNET Theta= 1
UNET Theta Warmup= 1
UNET ZTol= 0.006
UNET ZSATol= 0.006
UNET MxIter= 20
UNET Max Iter WO Improvement= 0
UNET MaxInSteps= 0
UNET DtIC= 0
UNET DtMin= 0
UNET MaxCRTS= 20
UNET WFStab= 2
UNET SFStab= 1
UNET WFX= 1
UNET SFX= 1
UNET 1D Methodology=Finite Difference
UNET DSS MLevel= 4
UNET Pardiso=0
UNET DZMax Abort= 30
UNET Use Existing IB Tables=-1
UNET Froude Reduction=False
UNET Froude Limit= 0.8
UNET Froude Power= 4
UNET D1 Cores= 0
UNET D2 Coriolis=0
UNET D2 Cores= 0
UNET D2 Theta= 1
UNET D2 Theta Warmup= 1
UNET D2 Z Tol= 0.003
UNET D2 Volume Tol= 0.003
UNET D2 Max Iterations= 20
UNET D2 Equation= 0
UNET D2 RampUpFraction=0.1
UNET D2 TimeSlices= 1
UNET D2 BCVolumeCheck=0
UNET D1D2 MaxIter= 0
UNET D1D2 ZTol=0.003
UNET D1D2 QTol=0.1
UNET D1D2 MinQTol=0.03
DSS File=dss
Write IC File= 0
Write IC File at Fixed DateTime=0
Write IC File at Sim End=0
Echo Input=False
Echo Parameters=False
Echo Output=False
Write Detailed= 0
HDF Write Warmup=0
HDF Write Time Slices=0
HDF Flush=0
HDF Face Node Velocities=0
HDF Compression= 1
HDF Chunk Size= 1
HDF Spatial Parts= 1
HDF Use Max Rows=0
HDF Fixed Rows= 1
Calibration Method= 0
Calibration Iterations= 20
Calibration Max Change=0.05
Calibration Tolerance=0.2
Calibration Maximum=1.5
Calibration Minimum=0.5
Calibration Optimization Method= 1
WQ AD Non Conservative
WQ ULTIMATE=-1
WQ Max Comp Step=1HOUR
WQ Output Interval=15MIN
WQ Output Selected Increments= 0
WQ Output face flow=0
WQ Output face velocity=0
WQ Output face area=0
WQ Output face dispersion=0
WQ Output cell volume=0
WQ Output cell surface area=0
WQ Output cell continuity=0
WQ Output cumulative cell continuity=0
WQ Output face conc=0
WQ Output face dconc_dx=0
WQ Output face courant=0
WQ Output face peclet=0
WQ Output face adv mass=0
WQ Output face disp mass=0
WQ Output cell mass=0
WQ Output cell source sink temp=0
WQ Output nsm pathways=0
WQ Output nsm derived pathways=0
WQ Output MaxMinRange=-1
WQ Daily Max Min Mean=-1
WQ Daily Range=0
WQ Daily Time=0
WQ Create Restart=0
WQ Fixed Restart=0
WQ System Summary=0
WQ Write To DSS=0
WQ Use Fixed Temperature=0
Sorting and Armoring Iterations= 10
XS Update Threshold= 0.02
Bed Roughness Predictor= 0
Hydraulics Update Threshold= 0.02
Energy Slope Method= 1
Volume Change Method= 1
Sediment Retention Method= 0
XS Weighting Method= 0
Number of US Weighted Cross Sections= 1
Number of DS Weighted Cross Sections= 1
Upstream XS Weight=0
Main XS Weight=1
Downstream XS Weight=0
Number of DS XS's Weighted with US Boundary= 1
Upstream Boundary Weight= 1
Weight of XSs Associated with US Boundary= 0
Number of US XS's Weighted with DS Boundary= 1
Downstream Boundary Weight= 0.5
Weight of XSs Associated with DS Boundary= 0.5
Percentile Method= 0
Sediment Output Level= 3
Mass or Volume Output= 0
Output Increment Type= 1
Profile and TS Output Increment= 1
XS Output Flag= 0
XS Output Increment= 10
Write Gradation File= 0
Read Gradation Hotstart= 0
Write HDF5 File= 1
Write Binary Output= 1
Write DSS Sediment File= 0
SV Curve= 0
Specific Gage Flag= 0

--- Stebenka.p01 (plan) ---

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Plan Title=ust_Q500
Short Identifier=ust_Q500
Geom File=g01
Flow File=u02
Computation Interval=2SEC
Run PostProcess= 0

--- Stebenka.p06 (plan) ---

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Plan Title=ust_Q100
Short Identifier=060521
Geom File=g04
Flow File=u03

--- Stebenka.p07 (plan) ---

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Plan Title=ust_Q20
Short Identifier=ust_Q20
Geom File=g04
Flow File=u04

--- Stebenka.f01 (steady flow) ---

Flow Title=Flow 01
Program Version=5.07
Number of Profiles= 1
Profile Names=PF 1
DSS Import GetInterval= 0
DSS Import GetPeak= 0
DSS Import FillOption= 0

--- Stebenka.u05 (unsteady flow) ---

Flow Title=ust_Q5
Program Version=5.07
Use Restart= 0
Restart Filename=Stebenka.p05.01SEP2008 0300_Q500.rst
Boundary Location=                ,                ,        ,        ,                ,Turnov          ,                ,HOP
Interval=1HOUR
Flow Hydrograph= 113
      14      14      14      14      14      14      14      14      14      14
      14      14      14      14      14      14      14      14      14      14
      14      14      14      14      14      14      14      14      14      14
      14      14      14      14      14      14      14      14      14      14
      14      14      14      14      14      14      14      14      14      14
      14      14      14      14      14      14      14      14      14      14
      14      14      14      14      14      14      14      14      14      14
      14      14      14      14      14      14      14      14      14      14
      14      14      14      14      14      14      14      14      14      14
      14      14      14      14      14      14      14      14      14      14
      14      14      14      14      14      14      14      14      14      14
      14      14      14
Stage Hydrograph TW Check=0
Flow Hydrograph Slope= 0.005
Use DSS=False
Use Fixed Start Time=False
Is Critical Boundary=False
Boundary Location=                ,                ,        ,        ,                ,Turnov          ,                ,DOP
Friction Slope=0.005,0

--- Stebenka.u01 (unsteady flow) ---

Flow Title=flow
Program Version=5.07
Use Restart= 0
Boundary Location=                ,                ,        ,        ,                ,Turnov          ,                ,HOP
Interval=1HOUR
Flow Hydrograph= 113
    44.6    44.6    44.6    44.6    44.6    44.6    44.6    44.6    44.6    44.6
    44.6    44.6    44.6    44.6    44.6    44.6    44.6    44.6    44.6    44.6
    44.6    44.6    44.6    44.6    44.6    44.6    44.6    44.6    44.6    44.6
    44.6    44.6    44.6    44.6    44.6    44.6    44.6    44.6    44.6    44.6
    44.6    44.6    44.6    44.6    44.6    44.6    44.6    44.6    44.6    44.6
    44.6    44.6    44.6    44.6    44.6    44.6    44.6    44.6    44.6    44.6
    44.6    44.6    44.6    44.6    44.6    44.6    44.6    44.6    44.6    44.6
    44.6    44.6    44.6    44.6    44.6    44.6    44.6    44.6    44.6    44.6
    44.6    44.6    44.6    44.6    44.6    44.6    44.6    44.6    44.6    44.6
    44.6    44.6    44.6    44.6    44.6    44.6    44.6    44.6    44.6    44.6
    44.6    44.6    44.6    44.6    44.6    44.6    44.6    44.6    44.6    44.6
    44.6    44.6    44.6
Stage Hydrograph TW Check=0
Use DSS=False
Use Fixed Start Time=False
Is Critical Boundary=False
Boundary Location=                ,                ,        ,        ,                ,Turnov          ,                ,DOP
Interval=1HOUR
Stage Hydrograph= 144
     248     248     248     248     248     248     248     248     248     248
     248     248     248     248     248     248     248     248     248     248
     248     248     248     248     248     248     248     248     248     248
     248     248     248     248     248     248     248     248     248     248
     248     248     248     248     248     248     248     248     248     248
     248     248     248     248     248     248     248     248     248     248
     248     248     248     248     248     248     248     248     248     248
     248     248     248     248     248     248     248     248     248     248
     248     248     248     248     248     248     248     248     248     248
     248     248     248     248     248     248     248     248     248     248
     248     248     248     248     248     248     248     248     248     248
     248     248     248     248     248     248     248     248     248     248
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Stage Hydrograph Use Initial Stage=-1
Stage Hydrograph TW Check=0
Use DSS=False
Use Fixed Start Time=False
Is Critical Boundary=False

--- Stebenka.u02 (unsteady flow) ---

Flow Title=ust_Q500
Program Version=5.07
Use Restart= 0
Restart Filename=Stebenka.p05.01SEP2008 0300_Q500.rst
Boundary Location=                ,                ,        ,        ,                ,Turnov          ,                ,HOP
Interval=1HOUR
Flow Hydrograph= 113
    44.6    44.6    44.6    44.6    44.6    44.6    44.6    44.6    44.6    44.6
    44.6    44.6    44.6    44.6    44.6    44.6    44.6    44.6    44.6    44.6
    44.6    44.6    44.6    44.6    44.6    44.6    44.6    44.6    44.6    44.6
    44.6    44.6    44.6    44.6    44.6    44.6    44.6    44.6    44.6    44.6
    44.6    44.6    44.6    44.6    44.6    44.6    44.6    44.6    44.6    44.6
    44.6    44.6    44.6    44.6    44.6    44.6    44.6    44.6    44.6    44.6
    44.6    44.6    44.6    44.6    44.6    44.6    44.6    44.6    44.6    44.6
    44.6    44.6    44.6    44.6    44.6    44.6    44.6    44.6    44.6    44.6
    44.6    44.6    44.6    44.6    44.6    44.6    44.6    44.6    44.6    44.6
    44.6    44.6    44.6    44.6    44.6    44.6    44.6    44.6    44.6    44.6
    44.6    44.6    44.6    44.6    44.6    44.6    44.6    44.6    44.6    44.6
    44.6    44.6    44.6
Stage Hydrograph TW Check=0
Flow Hydrograph Slope= 0.005
Use DSS=False
Use Fixed Start Time=False
Is Critical Boundary=False
Boundary Location=                ,                ,        ,        ,                ,Turnov          ,                ,DOP
Friction Slope=0.005,0

--- Stebenka.u03 (unsteady flow) ---

Flow Title=ust_Q100
Program Version=5.07
Use Restart= 0
Restart Filename=Stebenka.p05.01SEP2008 0300_Q500.rst
Boundary Location=                ,                ,        ,        ,                ,Turnov          ,                ,HOP
Interval=1HOUR
Flow Hydrograph= 113
    44.6    44.6    44.6    44.6    44.6    44.6    44.6    44.6    44.6    44.6
    44.6    44.6    44.6    44.6    44.6    44.6    44.6    44.6    44.6    44.6
    44.6    44.6    44.6    44.6    44.6    44.6    44.6    44.6    44.6    44.6
    44.6    44.6    44.6    44.6    44.6    44.6    44.6    44.6    44.6    44.6
    44.6    44.6    44.6    44.6    44.6    44.6    44.6    44.6    44.6    44.6
    44.6    44.6    44.6    44.6    44.6    44.6    44.6    44.6    44.6    44.6
    44.6    44.6    44.6    44.6    44.6    44.6    44.6    44.6    44.6    44.6
    44.6    44.6    44.6    44.6    44.6    44.6    44.6    44.6    44.6    44.6
    44.6    44.6    44.6    44.6    44.6    44.6    44.6    44.6    44.6    44.6
    44.6    44.6    44.6    44.6    44.6    44.6    44.6    44.6    44.6    44.6
    44.6    44.6    44.6    44.6    44.6    44.6    44.6    44.6    44.6    44.6
    44.6    44.6    44.6
Stage Hydrograph TW Check=0
Flow Hydrograph Slope= 0.005
Use DSS=False
Use Fixed Start Time=False
Is Critical Boundary=False
Boundary Location=                ,                ,        ,        ,                ,Turnov          ,                ,DOP
Friction Slope=0.005,0

--- Stebenka.u04 (unsteady flow) ---

Flow Title=ust_Q20
Program Version=5.07
Use Restart= 0
Restart Filename=Stebenka.p05.01SEP2008 0300_Q500.rst
Boundary Location=                ,                ,        ,        ,                ,Turnov          ,                ,HOP
Interval=1HOUR
Flow Hydrograph= 113
      22      22      22      22      22      22      22      22      22      22
      22      22      22      22      22      22      22      22      22      22
      22      22      22      22      22      22      22      22      22      22
      22      22      22      22      22      22      22      22      22      22
      22      22      22      22      22      22      22      22      22      22
      22      22      22      22      22      22      22      22      22      22
      22      22      22      22      22      22      22      22      22      22
      22      22      22      22      22      22      22      22      22      22
      22      22      22      22      22      22      22      22      22      22
      22      22      22      22      22      22      22      22      22      22
      22      22      22      22      22      22      22      22      22      22
      22      22      22
Stage Hydrograph TW Check=0
Flow Hydrograph Slope= 0.005
Use DSS=False
Use Fixed Start Time=False
Is Critical Boundary=False
Boundary Location=                ,                ,        ,        ,                ,Turnov          ,                ,DOP
Friction Slope=0.005,0

--- Stebenka.g04 (geometry) ---

Geom Title=Stebenka_objekty_2804
Program Version=5.07

Storage Area=Turnov          ,-683582.4880692,-995006.1043642
Storage Area Surface Line= 6
-684396.15111749-995363.99633007
-684234.40549412-994785.70710356
-683317.40572012-995063.49317766
-682610.70243561-994880.15043883
-684052.17550823-995055.42298498
-684396.15111749-995363.99633007
Storage Area Type= 1
Storage Area Is2D=-1
Storage Area Point Generation Data=0,0,3,3
Storage Area 2D Points= 37819
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Storage Area Mannings=0.06
2D Cell Volume Filter Tolerance=0.003
2D Cell Minimum Area Fraction=0.01
2D Face Profile Filter Tolerance=0.003
2D Face Area Elevation Profile Filter Tolerance=0.003
2D Face Area Elevation Conveyance Ratio=0.02
2D Face Area Laminar Depth=0.06

BreakLine Name=1
BreakLine Near Repeats=1
BreakLine Protection Radius=0
BreakLine Polyline= 2
-683668.69708312-995079.25863415 -683672.1030747-995091.36882641

BreakLine Name=m2
BreakLine Near Repeats=1
BreakLine Protection Radius=0
BreakLine Polyline= 4
-683888.27718101-995040.57459164 -683893.8065153-995045.97533676
-683897.53560122-995054.33363279 -683903.5792922-995060.76309127

BreakLine Name=M1
BreakLine Near Repeats=1
BreakLine Protection Radius=0
BreakLine Polyline= 4
-683949.25900695-995047.56096125-683951.23385113-995041.14271768
-683948.27158486-995028.60245716-683953.30743751-995020.30811162

BreakLine Name=M5
BreakLine Near Repeats=1
BreakLine Protection Radius=0
BreakLine Polyline= 4
-683499.96455115-995052.50862506-683502.72933495-995036.41363363
-683503.22304635-995023.67587968-683503.12430407-995008.86453788

BreakLine Name=lavka
BreakLine Near Repeats=1
BreakLine Protection Radius=0
BreakLine Polyline= 2
-683061.95532156 -994939.3827701-683067.02893792 -994927.0369703

Connection=lavka           ,-683064.4075695,-994933.8440723
Connection Line= 2
-683062.03988184-994939.67873106 -683066.7752571-994928.00941344
Conn CellSize Min=2
Conn CellSize Max=2
Conn Near Repeats=1
Conn Protection Radius=-1
Connection Up SA=Turnov
Connection Dn SA=Turnov
Conn Routing Type= 1
Conn Use RC Family=False
Conn OverFlow Method 2D=False
Conn Weir WD=1.3
Conn Weir Coef=1.66
Conn Weir Is Ogee= 0
Conn Simple Spill Pos Coef=0.05
Conn Simple Spill Neg Coef=0.05
Conn Weir SE= 7
       0 254.303    .567 254.385    .938 254.393   9.395 254.521   9.927  254.41
  11.092 254.672  12.594 254.894
Connection Culv=2,1.5,5,1.3,0.05,0.5,1,8,1,252.7,252.7, 1 ,Culvert #1  , 0 ,
     4.5     4.5
Conn Culvert Barrel=1,Barrel #1,0
Conn Culv Bottom n=0.25
Conn Outlet Rating Curve= 0 ,False,,

Connection=M               ,-683709.9963749,-995078.708676
Connection Line= 2
-683712.29585275-995082.94692939-683707.69689699-995074.47042268
Conn CellSize Min=1
Conn CellSize Max=1
Conn Near Repeats=1
Conn Protection Radius=-1
Connection Up SA=Turnov
Connection Dn SA=Turnov
Conn Routing Type= 1
Conn Use RC Family=False
Conn OverFlow Method 2D=False
Conn Weir WD=1.5
Conn Weir Coef=1.66
Conn Weir Is Ogee= 0
Conn Simple Spill Pos Coef=0.05
Conn Simple Spill Neg Coef=0.05
Conn Weir SE= 2
       0   249.2   9.644   249.2
Connection Culv=2,1.4,2.8,1.5,0.04,0.5,1,8,1,247.7,247.7, 1 ,Culvert #1  , 0 ,
     5.3     5.3
Conn Culvert Barrel=1,Barrel #1,0
Conn Culv Bottom n=0.04
Conn Outlet Rating Curve= 0 ,False,,

Connection=M1_sil.most     ,-683950.1993157,-995033.6564432
Connection Line= 4
-683949.16026474-995047.56096125-683951.23385113-995041.14271768
-683948.27158486-995028.70119937-683953.30743751-995020.40685383
Conn CellSize Min=3
Conn CellSize Max=3
Conn Near Repeats=1
Conn Protection Radius=-1
Connection Up SA=Turnov
Connection Dn SA=Turnov
Conn Routing Type= 1
Conn Use RC Family=False
Conn OverFlow Method 2D=False
Conn Weir WD=12.2
Conn Weir Coef=1.66
Conn Weir Is Ogee= 0
Conn Simple Spill Pos Coef=0.05
Conn Simple Spill Neg Coef=0.05
Conn Weir SE= 21
       0 249.269    .701  249.22   1.661 249.179    1.84 249.321   2.366 249.282
   2.891  249.27   4.993 249.326   5.518 249.306   6.044 249.257   6.355 249.272
   6.569 249.259   6.875 249.304   7.601 249.574   7.705  249.58  16.338 248.945
  16.852 248.915  18.394 248.967  19.534 248.962  25.191 248.844  26.812 248.742
  29.238 248.466
Connection Culv=2,2.7,6.7,12.2,0.04,0.5,1,8,1,245.72,245.72, 1 ,Culvert #1  , 0 ,
   12.22   12.22
Conn Culvert Barrel=1,Barrel #1,0
Conn Culv Bottom n=0.04
Conn Outlet Rating Curve= 0 ,False,,

Connection=M2_klenba       ,-683895.9756391,-995050.672931
Connection Line= 4
-683888.27718101-995040.70318081-683893.93510447-995046.10392593
-683897.66419039-995054.59081113 -683903.5792922-995060.76309127
Conn CellSize Min=1
Conn CellSize Max=1
Conn Near Repeats=1
Conn Protection Radius=-1
Connection Up SA=Turnov
Connection Dn SA=Turnov
Conn Routing Type= 1
Conn Use RC Family=False
Conn OverFlow Method 2D=False
Conn Weir WD=12.7
Conn Weir Coef=1.66
Conn Weir Is Ogee= 0
Conn Simple Spill Pos Coef=0.05
Conn Simple Spill Neg Coef=0.05
Conn Weir SE= 12
       0  248.99    3.64 249.045   6.535 249.148   7.396 249.227  17.421 249.522
  18.088 249.478  19.473 249.269  19.896 249.237  21.311 249.207  22.936 249.219
  23.171 249.259  25.641  249.31
Connection Culv=2,2.3,6.7,12.7,0.04,0.5,1,8,1,246.15,246.15, 1 ,Culvert #1  , 0 ,
    12.7    12.7
Conn Culvert Barrel=1,Barrel #1,0
Conn Culv Bottom n=0.04
Conn Outlet Rating Curve= 0 ,False,,

Connection=M5_U Strelnice  ,-683502.562523,-995031.0160125
Connection Line= 4
-683499.86580887-995052.70610961-683502.82807723-995036.41363363
-683503.42053091-995023.08342601-683503.51927318-995009.16076471
Conn CellSize Min=3
Conn CellSize Max=3
Conn Near Repeats=1
Conn Protection Radius=-1
Connection Up SA=Turnov
Connection Dn SA=Turnov
Conn Routing Type= 1
Conn Use RC Family=False
Conn OverFlow Method 2D=False
Conn Weir WD=40.77
Conn Weir Coef=1.66
Conn Weir Is Ogee= 0
Conn Simple Spill Pos Coef=0.05
Conn Simple Spill Neg Coef=0.05
Conn Weir SE= 21
       0 253.268   2.263 253.235   2.771 253.194   4.295 253.133   5.344 253.068
   7.853  252.89   8.026 252.845   9.042 252.771  11.129  252.56  12.599 252.456
  13.616 252.439  15.649 252.449  16.157 252.657  29.176 252.804  29.666 252.805
  30.006 252.539  35.507 252.536  37.507 252.555  40.007 252.602  42.007 252.667
  43.826 252.696
Connection Culv=6,2.9,,40.77,0.04,0.5,1,41,1,249.05,249.05, 1 ,Culvert #1  , 0 ,
    20.9    20.9
Conn Culvert Barrel=1,Barrel #2,0
Conn Culv Bottom n=0.04
Conn Outlet Rating Curve= 0 ,False,,

Connection=most            ,-683670.3527735,-995085.4556466
Connection Line= 2
-683671.96115838-995091.32152097-683668.74438856-995079.58977222
Conn CellSize Min=1
Conn CellSize Max=1
Conn Near Repeats=1
Conn Protection Radius=-1
Connection Up SA=Turnov
Connection Dn SA=Turnov
Conn Routing Type= 1
Conn Use RC Family=False
Conn OverFlow Method 2D=False
Conn Weir WD=2.6
Conn Weir Coef=1.66
Conn Weir Is Ogee= 0
Conn Simple Spill Pos Coef=0.05
Conn Simple Spill Neg Coef=0.05
Conn Weir SE= 10
       0 249.368     .53  249.37   3.123 249.418   3.641 249.445    4.16 249.513
   8.826 249.498   9.863 249.479  10.899 249.396  11.418  249.42  12.165 249.485
Connection Culv=2,1.7,3.2,2.6,0.04,0.5,1,8,1,247.65,247.65, 1 ,Culvert #1  , 0 ,
     6.6     6.6
Conn Culvert Barrel=1,Barrel #1,0
Conn Culv Bottom n=0.04
Conn Outlet Rating Curve= 0 ,False,,

BC Line Name=HOP
BC Line Storage Area=Turnov
BC Line Start Position=-682560.11084171 ,-994779.04472294
BC Line Middle Position=-682546.57993265 ,-994866.47521226
BC Line End Position=-682533.04902359 ,-994953.90570158
BC Line Arc= 2
-682560.11084171-994779.04472294-682533.04902359-994953.90570158

BC Line Name=DOP
BC Line Storage Area=Turnov
BC Line Start Position=-684406.84246936 ,-995362.27501239
BC Line Middle Position=-684316.303386575 ,-995395.09048781
BC Line End Position=-684225.76430379 ,-995427.90596323
BC Line Arc= 2
-684406.84246936-995362.27501239-684225.76430379-995427.90596323
LCMann Table=5
budova,5
les,0.08
voda,0.035
zelen? plocha,0.06
zpevnen? plocha,0.025

Chan Stop Cuts=-1
Use User Specified Reach Order=0
Composite Channel Slope=5
